HEC-RAS study LAURELRN1.prj: LAURELRN1

--- LAURELRN1.g01 (geometry) --- (continued)

Type RM Length L Ch R = 1 ,27782   ,367.7,369.4,370.9
XS GIS Cut Line= 3
2214569.09951041391831.160755166 2214396.8179759392295.016167345
2214334.31607315392395.426567144
#Sta/Elev= 30
       0 2523.72    19.2 2512.28    49.1 2496.87    83.2 2477.89   100.3 2468.94
   117.4 2461.76   134.4 2449.61     143 2440.45     160 2426.67   164.3 2425.45
   181.4 2425.96   195.2 2423.34   211.2 2422.18     224 2423.26   263.6 2426.76
   279.2 2425.82   305.1 2426.84   316.5 2425.98   332.1 2426.24   344.5 2425.15
   394.7 2424.82   407.5 2427.05   444.1 2426.09   475.8 2426.66   484.6 2429.64
   505.6 2440.16   534.6 2456.71   549.5 2463.47     568 2474.09   613.1 2497.18
#Mann= 5 ,-1,0
       0      .1       0     120     .12       0   195.2    .045       0
     224     .12       0     330      .1       0
#XS Ineff= 2 , 0
                          466.28         2446.05
Permanent Ineff=
       F       F
Bank Sta=195.2,224
XS Rating Curve= 0 ,0
Exp/Cntr(USF)=0,0
Exp/Cntr=0.3,0.1

Type RM Length L Ch R = 1 ,27412   ,541.6,545.3,538.8
XS GIS Cut Line= 2
 2214232.1627747391747.3147082952214017.02749821392155.388764497
#Sta/Elev= 30
       0 2491.48    15.7 2484.43    36.9 2473.09    56.4 2463.78    63.5 2459.57
    74.5 2454.05      88 2442.88   106.1 2426.65   110.9 2421.65   115.2  2419.1
   141.22419.319   146.8 2420.27   160.4 2421.41   178.5 2421.19   199.7 2422.56
   210.1 2421.45   223.4 2422.71   270.8 2422.35   282.5 2423.05     296 2422.06
   314.1 2421.88   325.9 2421.09   359.3 2421.08     391 2418.77   395.2 2419.12
     400  2422.3   411.7 2432.48   436.6 2455.26   445.2  2460.7   461.3 2469.71
#Mann= 5 ,-1,0
       0      .1       0     110     .12       0   115.2    .045       0
   141.2     .12       0     240      .1       0
#XS Ineff= 2 , 0
                           380.4         2438.54
Permanent Ineff=
       F       F
Bank Sta=115.2,141.2
XS Rating Curve= 0 ,0
Exp/Cntr(USF)=0,0
Exp/Cntr=0.3,0.1

Type RM Length L Ch R = 1 ,26867   ,436.6,431.5,416.6
XS GIS Cut Line= 2
2213827.50356416391479.249324095 2213614.0757105391919.764414054
#Sta/Elev= 30
       0 2496.72    33.3 2481.54    46.6 2474.27    78.8 2453.15    87.8 2446.08
    99.7 2434.61   108.5 2427.05   117.7 2420.84   123.7 2417.94   132.7 2417.08
   162.2 2418.87   172.8 2416.44   179.9 2415.68   184.4 2415.83   193.3  2417.6
   237.7 2417.77   259.9 2417.17   268.8 2416.19   326.6 2416.65   339.9 2416.03
   384.4 2415.75   390.2  2415.2   402.1 2413.63   411.1  2414.4   415.5  2415.4
     420 2419.18   433.3 2434.32   442.2 2442.46     459  2453.3   489.5 2471.52
#Mann= 5 ,-1,0
       0      .1       0     190     .12       0     300      .1       0
   390.2    .045       0   415.5      .1       0
#XS Ineff= 2 , 0
          158.22 2436.65
Permanent Ineff=
       F       F
Bank Sta=390.2,415.5
XS Rating Curve= 0 ,0
Exp/Cntr(USF)=0,0
Exp/Cntr=0.3,0.1

Type RM Length L Ch R = 1 ,26435   ,549.5,548.2,538.6
XS GIS Cut Line= 4
2213289.66537293391399.0004511182213238.44268805391530.472008974
2213289.66537293391841.2229639062213400.64785684392088.799274154
#Sta/Elev= 30
       0 2452.85    19.5 2444.35    53.9 2422.12    66.7  2417.3    79.6  2416.1
   120.2 2416.69   200.6 2410.56   208.7  2412.2     229 2412.72   245.2 2410.88
   265.5 2412.03   281.7 2411.22   293.8 2412.94   301.6 2411.27     306 2409.93
   321.82411.368   358.7 2409.82   399.2 2412.69   433.8 2411.57   440.8 2413.27
   451.9 2418.96   477.9 2436.34     560 2479.63   653.3  2539.4   663.7 2544.49
   666.8 2546.76   670.8 2551.62   679.6 2558.34     697 2573.84   727.4  2588.9
#Mann= 5 ,-1,0
       0      .1       0      60     .12       0   301.6    .045       0
   321.8     .12       0   361.1      .1       0
Bank Sta=301.6,321.8
XS Rating Curve= 0 ,0
Exp/Cntr(USF)=0,0
Exp/Cntr=0.3,0.1

Type RM Length L Ch R = 1 ,25887   ,528.5,531.5,532.3
XS GIS Cut Line= 3
2212693.77480551391554.3759285842212785.97563829391648.284184196
 2213007.9406061392059.773086056
#Sta/Elev= 30
       0 2483.76     9.5 2473.62    51.8 2443.18    65.9 2431.43    77.6 2423.33
      88 2417.74    94.2 2416.03   121.6 2412.42   154.6  2409.3   172.3 2405.69
   184.1 2405.94   191.7 2406.94   254.9 2406.69   264.4 2407.64   287.1 2406.03
     314 2407.75   349.4 2407.27   363.7  2408.2   370.1 2407.95   380.6 2405.05
   405.5 2406.46   437.1 2405.55   470.5 2407.17   508.8 2405.68   518.9 2406.79
   523.6 2410.09   542.8 2429.07   564.9  2446.4   576.7 2454.13   599.1 2465.02
#Mann= 5 ,-1,0
       0      .1       0   172.3    .045       0   184.1      .1       0
   251.6     .12       0   471.6      .1       0
#XS Ineff= 2 , 0
                          457.14         2420.07
Permanent Ineff=
       F       F
Bank Sta=172.3,184.1
XS Rating Curve= 0 ,0
Exp/Cntr(USF)=0,0
Exp/Cntr=0.3,0.1

Type RM Length L Ch R = 1 ,25356   ,348.6,351.3,352.2
XS GIS Cut Line= 2
2212388.14611906391912.9347227372212666.45604024392351.742389866
#Sta/Elev= 30
       0 2425.85    19.2 2417.55    42.9 2409.76    67.3 2404.88    90.3 2403.37
   104.5 2403.69   112.1 2400.73   118.7  2400.1   142.2 2400.82     185 2400.44
   194.2 2399.05     204 2397.64   220.5 2398.83   232.4 2402.67   246.5 2403.47
   307.4 2401.02   321.2 2401.31   327.7  2400.6   350.9 2400.47   365.4 2399.63
   379.2 2400.69   382.8 2402.56   385.7 2404.88   403.3 2422.89   407.6 2426.39
   449.4 2456.56   455.2 2460.17   464.5 2464.55   487.1 2478.39   519.6 2496.16
#Mann= 5 ,-1,0
       0      .1       0     160     .12       0   194.2    .045       0
   220.5     .12       0     300      .1       0
#XS Ineff= 2 , 0
                          328.11         2424.42
Permanent Ineff=
       F       F
Bank Sta=194.2,220.5
XS Rating Curve= 0 ,0
Exp/Cntr(USF)=0,0
Exp/Cntr=0.3,0.1

Type RM Length L Ch R = 1 ,25004   ,289.6,286.3,281.9
XS GIS Cut Line= 3
2212113.25104355392081.9695828372212290.82301779392445.650645477
2212410.34261584392582.244471821
#Sta/Elev= 30
       0 2469.05    30.3 2449.05    46.5 2435.62      57 2428.39    83.7 2411.26
    97.8 2403.37   106.9 2399.71   114.9 2398.11   134.3 2398.02   159.4 2399.88
   172.7 2395.54   181.1 2394.66     195  2395.3   207.2 2394.34   230.6 2396.55
   243.9 2395.59   257.3 2396.55   279.6 2396.07   306.3 2398.47   337.4 2398.49
   350.8 2396.91   375.5  2398.9   406.8 2398.72   439.4 2402.84   451.9 2408.39
   473.4 2422.26     510 2453.39   535.7 2472.99   563.5 2489.34   586.2 2500.96
#Mann= 4 ,-1,0
       0      .1       0   172.7    .045       0     195     .12       0
  504.72      .1       0
#XS Ineff= 2 , 0
                          390.78         2421.51
Permanent Ineff=
       F       F
Bank Sta=172.7,195
XS Rating Curve= 0 ,0
Exp/Cntr(USF)=0,0
Exp/Cntr=0.3,0.1

Type RM Length L Ch R = 1 ,24718   ,251.3,252.4,254
XS GIS Cut Line= 3
2211881.40729159392315.7581805332212028.24565491392488.207886292
 2212243.3809314392645.290786587
#Sta/Elev= 30
       0    2453    12.4  2447.7    39.9 2432.62    53.6 2423.98    75.4 2411.43
    96.4 2398.52     103 2397.89   109.2 2395.94   117.4  2391.1   121.5 2390.58
   133.2  2390.5     142 2391.25   150.5 2392.81   164.7 2394.56   196.2 2395.94
   220.2 2395.68   236.3 2396.37   246.2 2395.94   280.9 2396.12   316.3  2397.5
     396 2397.05   418.1 2397.53   424.9 2396.72   429.5 2396.78   433.2 2398.42
   436.1 2400.53   450.4  2413.7   469.1 2428.21   487.6 2441.03   492.9 2444.29
#Mann= 4 ,-1,0
       0      .1       0   117.4    .045       0     142     .12       0
   476.5      .1       0
#XS Ineff= 2 , 0
                          278.35         2403.86
Permanent Ineff=
       F       F
Bank Sta=117.4,142
XS Rating Curve= 0 ,0
Exp/Cntr(USF)=0,0
Exp/Cntr=0.3,0.1

Type RM Length L Ch R = 1 ,24466   ,482.9,474.7,471.7
XS GIS Cut Line= 4
2211676.51655208392431.8629329252211871.16275462392717.002545417
2211848.96625783392872.3780228832211920.67801666393027.753500349
#Sta/Elev= 30
       0 2452.23    30.7 2439.62    56.2 2426.39    83.9 2409.65    98.5 2398.22
   108.1 2391.94   112.9 2391.16   127.1 2391.69   153.3 2390.76   166.3 2389.95
   173.4 2388.53   183.9 2387.78   193.5 2388.85     205 2392.62   219.3 2391.16
   248.6 2391.92   276.1 2390.27     297 2391.06   311.5 2392.81   349.5 2393.87
   358.6 2393.02   446.4 2391.48   494.9 2393.44     578 2398.72     600 2401.21
   608.8 2403.23   622.8 2408.95   639.6 2418.07   644.1 2419.31   673.3 2423.27
#Mann= 5 ,-1,0
       0      .1       0   173.4    .045       0   193.5      .1       0
     250     .12       0  465.24      .1       0
#XS Ineff= 2 , 0
                          347.44         2410.31
Permanent Ineff=
       F       F
Bank Sta=173.4,193.5
XS Rating Curve= 0 ,0
Exp/Cntr(USF)=0,0
Exp/Cntr=0.3,0.1

Type RM Length L Ch R = 1 ,23991   ,313.6,315.3,314.6
XS GIS Cut Line= 2
2211331.61714056 392662.365014882211801.15841861393029.460923179
#Sta/Elev= 30
       0 2444.48    24.1 2427.33    46.4  2407.5    51.5 2402.29    62.2 2388.15
    65.1 2385.59    67.9 2384.87      89  2385.5   107.3 2388.46   140.9 2387.21
   153.9 2388.18   184.8 2388.32   199.4 2387.49   205.9 2385.58   212.4 2385.06
   224.1 2385.89   230.4  2388.5   236.1 2389.13   273.1  2388.9     285 2387.74
   303.3 2389.52   335.8 2389.91   367.1 2388.53   417.1 2388.69   441.2 2387.63
   452.7 2389.32   492.5 2390.43   523.9 2393.92   572.3 2404.46     596 2408.62
#Mann= 5 ,-1,0
       0      .1       0    65.1    .045       0      89      .1       0
     180     .12       0     430      .1       0
#XS Ineff= 2 , 0
                          416.59         2401.92
Permanent Ineff=
       F       F
Bank Sta=65.1,89
XS Rating Curve= 0 ,0
Exp/Cntr(USF)=0,0
Exp/Cntr=0.3,0.1

Type RM Length L Ch R = 1 ,23676   ,495.9,497.5,494.3
XS GIS Cut Line= 3
2211113.06701841392874.0854457132211452.84416144393155.810212547
2211556.99695402393256.548159475
#Sta/Elev= 30
       0 2446.52    11.1 2442.34    61.2 2419.83    66.4 2415.81    83.9 2399.92
    89.6 2396.32    98.1 2392.25   118.4 2387.05   133.9 2382.14   143.6 2382.01
   149.5 2382.89   154.7 2382.22   165.1 2381.28   172.72382.187   191.9 2384.25
   217.9 2384.18   232.7 2382.52   261.8 2383.39   274.3 2385.03   355.8 2383.26
   368.3 2381.32   378.2 2383.26   399.7 2384.64   430.5 2388.82   449.1 2387.51
   489.4 2387.97   496.1 2388.98   512.8 2394.04   552.2  2410.8   586.3 2418.05
#Mann= 7 ,-1,0
       0      .1       0   154.7    .045       0   172.7      .1       0
     340     .12       0     400      .1       0  461.38     .12       0
  541.38      .1       0
#XS Ineff= 2 , 0
                          432.68         2391.77
Permanent Ineff=
       F       F
Bank Sta=154.7,172.7
XS Rating Curve= 0 ,0
Exp/Cntr(USF)=0,0
Exp/Cntr=0.3,0.1

Type RM Length L Ch R = 1 ,23178   ,259.4,260.3,260
XS GIS Cut Line= 2
2210896.22431909393184.8364006452211271.85734153393569.006537236
#Sta/Elev= 30
       0 2416.16    17.3 2405.55    39.6 2386.39    45.2    2383    50.8 2381.02
      54 2380.45   116.2 2381.09   133.2 2379.06   147.3 2379.74   160.1 2378.95
   181.2 2380.62   189.7 2380.27   201.9 2380.93     218 2380.47   237.8 2381.46
     246 2381.25   257.6 2378.78   308.5 2379.87   314.2 2379.38   322.7  2377.7
   330.5 2377.38     334 2377.68   352.9 2381.54   377.5 2385.56   453.6 2385.55
   487.2 2386.84   509.6  2388.9   526.3 2393.77     532 2395.88   537.3 2398.45
#Mann= 6 ,-1,0
       0      .1       0     260     .12       0   322.7    .045       0
     334      .1       0     400     .12       0     470      .1       0
#XS Ineff= 2 , 0
          107.83 2391.18
Permanent Ineff=
       F       F
Bank Sta=322.7,334
XS Rating Curve= 0 ,0
Exp/Cntr(USF)=0,0
Exp/Cntr=0.3,0.1

Type RM Length L Ch R = 1 ,22918   ,492.7,505.7,507
XS GIS Cut Line= 2
2210677.67419694393336.7970324522211092.57794446393744.871088654
#Sta/Elev= 30
       0 2420.92     7.7 2414.46    21.8 2401.04    38.8 2385.99    46.2 2380.77
    51.9 2378.68    67.1 2378.04    82.1 2376.32    98.9 2376.82     118 2376.33
   138.2 2377.32     166 2376.25   205.7 2376.32   216.7 2376.92   250.9 2375.38
   268.7 2375.78     284 2378.05     320 2378.89   345.7 2377.86   366.9 2375.75
   396.2 2375.67   434.8 2380.69   463.1 2381.22     497 2385.08   525.3 2386.62
   542.5 2389.47   553.6 2392.17   567.7  2398.3   575.8  2400.3     582  2403.6
#Mann= 5 ,-1,0
       0      .1       0     280     .12       0   366.9    .045       0
   396.2     .12       0     540      .1       0
#XS Ineff= 2 , 0
           88.48 2394.97
Permanent Ineff=
       F       F
Bank Sta=366.9,396.2
XS Rating Curve= 0 ,0
Exp/Cntr(USF)=0,0
Exp/Cntr=0.3,0.1

Type RM Length L Ch R = 1 ,22412   ,407,406.4,404.4
XS GIS Cut Line= 3
 2210465.9537661393661.207370018 2210664.0148143 393997.56966739
2210756.21564709394088.063077342
#Sta/Elev= 30
       0 2410.79    27.8 2405.54    60.3 2400.65      65 2399.35    75.3 2389.75
    83.4 2383.77   106.7 2372.87   122.6 2371.61   133.1 2371.22   139.2 2371.47
   148.5 2373.03   157.8 2372.52   194.9 2372.89   208.9 2372.39   222.8 2373.54
   229.5 2373.39   240.9 2374.77   279.2 2373.89   299.6 2371.31   338.8 2373.56
   357.4 2372.99     376 2376.89   407.2 2379.62   424.2 2381.85   441.2 2385.15
   458.1 2389.47   469.7 2393.82   481.2 2396.83   503.3 2404.49   519.5 2408.85
#Mann= 7 ,-1,0
       0      .1       0   122.6    .045       0   139.2      .1       0
     180     .12       0     230      .1       0     290     .12       0
  420.34      .1       0
Bank Sta=122.6,139.2
XS Rating Curve= 0 ,0
Exp/Cntr(USF)=0,0
Exp/Cntr=0.3,0.1

Type RM Length L Ch R = 1 ,22006   ,390,390.1,378.5
XS GIS Cut Line= 3
2210148.37311986393917.3207944132210402.77912142394246.853400467
2210522.29871947394356.128461542
#Sta/Elev= 30
       0 2404.34    38.9 2377.03      52 2370.83    68.2 2369.24    76.8 2369.61
    88.2 2367.51   125.2 2369.94   143.7 2368.99   156.5 2368.31   170.9 2368.86
   202.6 2368.02   217.1 2368.52   227.9 2366.27   236.5 2368.62   241.9  2369.2
   282.8 2369.03   292.9 2366.91   299.2 2367.31   310.6 2366.37   323.2 2367.83
   358.6 2368.75   373.8 2366.19   384.7  2368.6   418.2 2370.34   443.5 2372.73
   472.4 2377.15   483.2 2380.16   504.9 2389.45   542.9 2395.96   578.3 2408.92
#Mann= 3 ,-1,0
       0      .1       0   143.7    .045       0   170.9      .1       0
Bank Sta=143.7,170.9
XS Rating Curve= 0 ,0
Exp/Cntr(USF)=0,0
Exp/Cntr=0.3,0.1

Type RM Length L Ch R = 1 ,21616   ,179.6,179.3,178.6
XS GIS Cut Line= 2
2209928.76496307394158.3802742782210207.07488425394477.668343356
#Sta/Elev= 30
       0 2399.96     5.2 2398.33    14.3 2394.19    30.2 2384.75    49.8 2374.92
    63.9 2366.04    72.4  2363.7    84.3 2362.67    88.6 2363.19    93.9 2365.61
    96.5 2366.06   109.3 2365.62   131.1 2366.44     183 2366.63   191.5 2365.54
   210.7 2364.77   273.7  2365.7   285.1 2364.51   291.3 2362.17   307.8 2361.28
   313.4 2360.91   321.7 2361.24     338    2362   341.8 2363.75   346.1 2366.49
   352.2 2371.64   369.8 2388.92   375.8 2393.54   380.5 2395.74   423.6 2402.86
#Mann= 3 ,-1,0
       0      .1       0   307.8    .045       0   321.7      .1       0
#XS Ineff= 2 , 0
            93.7 2375.01
Permanent Ineff=
       F       F
Bank Sta=307.8,321.7
XS Rating Curve= 0 ,0
Exp/Cntr(USF)=0,0
Exp/Cntr=0.3,0.1

Type RM Length L Ch R = 1 ,21436   ,273.7,270.4,268.4
XS GIS Cut Line= 3
  2209844.511464394297.3735670892210036.75020035394555.996903042
2210093.45371251394601.636315269
#Sta/Elev= 30
       0 2386.41    11.1 2384.04    16.8 2381.85    24.7 2377.47    33.9 2370.58
    39.7 2367.08    49.6 2363.36    84.5 2361.64    96.8 2362.83   119.4 2363.15
   140.2 2363.22   179.2 2361.84     194 2362.75   199.1 2361.54   202.32360.146
   209.1 2359.17     229 2360.04     234 2361.06     249 2361.85   274.1 2360.87
   278.9  2361.6   282.7 2363.85   287.8 2367.79   299.8 2379.28   305.5 2382.67
   311.2  2384.8   326.6 2388.63     342 2391.13   368.8 2395.21     395 2398.14
#Mann= 3 ,-1,0
       0      .1       0   202.3    .045       0     229      .1       0
#XS Ineff= 2 , 0
           83.56 2372.47
Permanent Ineff=
       F       F
Bank Sta=202.3,229
XS Rating Curve= 0 ,0
Exp/Cntr(USF)=0,0
Exp/Cntr=0.3,0.1

Type RM Length L Ch R = 1 ,21166   ,339.6,341.5,342.2
XS GIS Cut Line= 3
2209613.54837788394490.9953159312209847.27748898394719.192377066
2209937.17330095394788.343001653
#Sta/Elev= 30
       0 2396.16      26 2384.66    48.7 2378.44    54.7 2374.66    65.6 2365.39
    71.8 2361.13    76.3  2358.7    81.9 2357.42    96.7 2357.27   108.1 2359.11
   122.2 2358.02   136.3 2358.41     152 2356.75   173.1  2359.9   180.6 2360.31
   199.3 2359.47     224 2359.97   235.3 2357.93   249.5 2359.74     272 2357.42
   289.4 2357.71   300.4 2356.49   303.2 2357.55   308.9 2361.05   320.2 2364.97
     343 2366.91   363.1 2367.17   377.2 2370.86   398.4  2377.7   440.1  2383.7
#Mann= 3 ,-1,0
       0      .1       0     272    .045       0   303.2      .1       0
Bank Sta=272,303.2
XS Rating Curve= 0 ,0
Exp/Cntr(USF)=0,0
Exp/Cntr=0.3,0.1

Type RM Length L Ch R = 1 ,20824   ,262.6,261.9,258.1
XS GIS Cut Line= 3
 2209359.0740794394679.0850148062209570.67499064394912.814125908
 2209660.5708026395131.330099602
#Sta/Elev= 30
       0  2412.3    40.6 2389.69    64.6 2379.53    78.7 2376.02    92.9 2373.56
   108.9  2372.3   132.5 2367.61   143.9 2367.33     158 2363.64   172.2 2356.98
   186.3    2355     192 2353.25   197.1 2353.09   213.3 2355.39   234.5 2355.46
   245.62353.789     260 2353.14   268.5 2353.96   272.6 2355.28   285.5 2355.71
   311.6 2358.89   356.6 2360.07   368.8 2364.88   384.9  2374.1   408.6    2389
   419.5 2394.06   445.4 2397.47   501.7 2402.46   536.3 2407.34   551.6 2410.31
#Mann= 3 ,-1,0
       0      .1       0   245.6    .045       0   268.5      .1       0
Bank Sta=245.6,268.5
XS Rating Curve= 0 ,0
Exp/Cntr(USF)=0,0
Exp/Cntr=0.3,0.1

Type RM Length L Ch R = 1 ,20563   ,179.7,186.3,189.7
XS GIS Cut Line= 4
 2209197.8202204394871.4042937072209287.43942987 394984.67301678
2209495.30620738395158.932590738 2209516.4662985395190.050371802
#Sta/Elev= 30
       0 2380.96    27.8 2367.57    48.2 2356.55    53.3 2354.79    68.6  2354.9
    96.9 2353.06   150.6 2354.97   155.8 2354.28   162.4 2352.38   181.9 2351.97
  189.67 2350.37     195 2349.84   219.9 2350.32   239.3 2350.59   249.8 2352.22
   287.3 2354.03   294.7 2353.63   304.3 2351.84   319.6 2353.43   335.6 2351.95
   344.5 2351.86     349 2353.22   359.4 2360.06   369.8 2367.74   381.8 2378.01
     388 2382.22     413 2387.75   432.9 2393.42   442.6 2396.72   453.3 2401.46
#Mann= 3 ,-1,0
       0      .1       0  189.67    .045       0   219.9      .1       0
#XS Ineff= 2 , 0
           68.36 2367.33  323.35         2367.59
Permanent Ineff=
       F       F
Bank Sta=189.67,219.9
XS Rating Curve= 0 ,0
Exp/Cntr(USF)=0,0
Exp/Cntr=0.3,0.1

Type RM Length L Ch R = 1 ,20376   ,140,139.8,138.9
XS GIS Cut Line= 3
2209047.60760178394932.5058088372209290.83345468395269.954289428
2209348.90088802395309.396319627
#Sta/Elev= 30
       0  2393.5    12.4 2388.03    20.9 2382.58    35.3 2375.32    63.9 2357.19
    72.5 2353.37    99.4  2350.1   109.3 2350.33   124.1 2352.31     134 2352.27
   155.6 2347.94   172.8 2350.07   184.3 2349.11   206.2 2350.82   221.5 2350.61
   242.4 2351.79   264.5 2351.28   274.6 2348.41   300.7  2348.4   311.5 2349.12
   322.5 2351.14   331.2 2350.45   350.9 2351.34   360.8 2348.38   390.6 2349.62
   399.2  2352.3   404.6 2355.14   421.7 2368.49   432.1 2374.09   486.2 2396.51
#Mann= 3 ,-1,0
       0      .1       0   274.6    .045       0   300.7      .1       0
#XS Ineff= 2 , 0
          132.87 2364.09
Permanent Ineff=
       F       F
Bank Sta=274.6,300.7
XS Rating Curve= 0 ,0
Exp/Cntr(USF)=0,0
Exp/Cntr=0.3,0.1

Type RM Length L Ch R = 1 ,20236   ,277.3,291.4,296.6
XS GIS Cut Line= 2
2208937.67557071395022.0143540562209187.86253046395353.107544577
#Sta/Elev= 30
       0 2395.45      19 2390.41      24 2388.91    26.9 2387.42    46.9 2372.72
    69.1  2354.7    77.1 2348.84    84.2 2345.72    94.2 2345.49   118.3  2346.9
   163.4 2347.91   174.4 2349.67   189.5 2348.23   216.5 2350.48   241.1 2349.98
   266.8 2348.52   284.7 2346.85   306.7 2346.08   309.6 2346.11   311.2 2346.75
   315.3 2348.82     321 2350.54   324.8 2350.77   335.3 2349.52   359.9 2350.83
   369.1 2354.83     390 2366.94   398.1 2371.06   403.8 2373.24     415 2375.75
#Mann= 3 ,-1,0
       0      .1       0   284.7    .045       0   311.2      .1       0
#XS Ineff= 2 , 0
           95.24 2361.99  355.61         2364.42
Permanent Ineff=
       F       F
Bank Sta=284.7,311.2
XS Rating Curve= 0 ,0
Exp/Cntr(USF)=0,0
Exp/Cntr=0.3,0.1

Type RM Length L Ch R = 1 ,19945   ,223.1,215,206.8
XS GIS Cut Line= 5
2208843.82377909395037.6845560342208881.07458539395161.488706381
2208952.28936213395249.1376623792208965.43670553395376.228648576
2209004.87873573395461.686380673
#Sta/Elev= 30
       0 2405.79      12  2400.5    37.1 2387.76    54.5 2380.13    66.3 2375.62
    70.5 2373.51    87.2 2359.41      93 2355.89  113.49    2345   116.4 2343.99
   125.1 2344.97   139.2 2344.83     165 2345.85   185.3 2345.24     201 2346.79
   213.7 2346.99   233.6 2349.04   242.2 2349.04   258.3 2348.08   298.6 2348.97
   322.7 2350.35   342.8 2352.19   354.5 2354.26     371 2358.29   393.1 2365.87
     412 2371.55   432.7 2377.09   441.5 2379.93   451.1  2382.4   464.1  2385.1
#Mann= 3 ,-1,0
       0      .1       0  113.49    .045       0   125.1      .1       0
#XS Ineff= 2 , 0
                          293.39         2360.11
Permanent Ineff=
       F       F
Bank Sta=113.49,125.1
XS Rating Curve= 0 ,0
Exp/Cntr(USF)=0,0
Exp/Cntr=0.3,0.1

Type RM Length L Ch R = 1 ,19730   ,176.1,179,178.8
XS GIS Cut Line= 3
2208670.33385852395228.1409740232208793.42197029395323.568835952
2208923.42514451395482.615272501
#Sta/Elev= 30
       0 2375.89    22.6 2367.53    27.6 2364.37    42.8 2351.75    52.9 2345.76
      58 2343.24    61.9 2342.05    73.3 2342.91    78.2 2342.58    88.4 2340.84
    93.1 2340.68   100.52341.118   116.1 2341.07   133.2 2341.84     136 2342.55
     144 2346.48   149.1 2347.12   167.4 2347.49   183.7 2346.32   204.3 2347.44
   240.5 2350.65   254.9 2350.36   266.9  2350.8   286.8    2353   295.3 2355.05
   306.7 2359.64   330.7 2372.69   343.8 2378.99   349.7 2381.02   361.2 2382.32
#Mann= 3 ,-1,0
       0      .1       0   100.5    .045       0   116.1      .1       0
#XS Ineff= 2 , 0
                          164.73         2349.55
Permanent Ineff=
       F       F
Bank Sta=100.5,116.1
XS Rating Curve= 0 ,0
Exp/Cntr(USF)=0,0
Exp/Cntr=0.3,0.1

Type RM Length L Ch R = 1 ,19551   ,216.2,216.7,216.8
XS GIS Cut Line= 3
2208558.03864173395343.1498546362208713.62754705395488.781070016
2208792.04435533395564.708455812
#Sta/Elev= 30
       0 2371.63    11.4 2365.44    17.1 2362.69    30.3 2357.27    41.3 2353.19
    45.4 2350.91    52.2 2346.06    59.5 2341.71    65.2 2339.01    67.4  2338.3
    74.2 2337.92    79.4 2337.97    82.2 2338.46    90.6 2340.39    96.1 2340.62
   114.2 2339.61   124.6 2339.71   133.1 2338.81   137.6 2338.73   155.2    2339
   169.9 2340.44   186.9 2340.96   192.6  2341.6     202 2344.26   209.5 2345.51
   232.2 2346.57   274.6 2349.97   305.7 2356.31     317 2357.87   322.3 2358.24
#Mann= 3 ,-1,0
       0      .1       0    67.4    .045       0    82.2      .1       0
Bank Sta=67.4,82.2
XS Rating Curve= 0 ,0
Exp/Cntr(USF)=0,0
Exp/Cntr=0.3,0.1

Type RM Length L Ch R = 1 ,19334   ,236.7,233.4,230.2
XS GIS Cut Line= 2
2208386.26849026395472.5998238622208652.63669616395736.478607285
#Sta/Elev= 30
       0 2387.37     6.5 2382.87    15.9 2375.21    25.2 2369.14    32.9 2363.46
    42.1 2356.19      59 2344.73    63.3 2342.28    70.2  2339.5    86.72335.081
    98.4 2334.68   106.4 2335.04   134.7 2336.27   148.8 2337.86     163 2338.55
     180 2337.42   194.1 2338.25   211.1 2338.28     228 2335.73   233.7  2335.6
   236.5 2336.32   245.2 2340.39   273.6 2341.14   302.1 2340.13   306.7 2340.72
   318.5  2345.5   323.6 2346.34   335.5 2346.88     344 2346.56   374.9 2347.77
#Mann= 3 ,-1,0
       0      .1       0    86.7    .045       0   106.4      .1       0
#XS Ineff= 2 , 0
                          249.69         2343.95
Permanent Ineff=
       F       F
Bank Sta=86.7,106.4
XS Rating Curve= 0 ,0
Exp/Cntr(USF)=0,0
Exp/Cntr=0.3,0.1

Type RM Length L Ch R = 1 ,19101   ,209.6,207.7,205
XS GIS Cut Line= 4
2208215.74305003395630.6781516672208254.32909855395680.466601369
2208398.71560268395775.0646558042208529.41028315395849.747330357
#Sta/Elev= 30
       0 2365.19    16.3 2353.37    27.7  2344.4    33.5 2340.76    38.6 2338.51
    47.7 2337.09    53.4 2336.88    73.5 2338.47    79.5 2338.13    94.7 2331.79
   108.2 2331.25   116.8 2331.81   136.9 2333.76   156.1 2334.12   180.4 2336.03
   184.7 2335.75   189.5 2333.77   194.3 2332.74   197.7 2332.88   203.9 2333.97
   213.4 2337.33   226.6 2338.33     247 2338.61   273.4  2336.3   305.7 2337.72
   317.4 2337.13   320.5 2337.38     334 2342.08   368.9 2345.36   386.1 2348.44
#Mann= 3 ,-1,0
       0      .1       0    94.7    .045       0   116.8      .1       0
#XS Ineff= 2 , 0
           74.59  2343.1  234.37         2341.35
Permanent Ineff=
       F       F
Bank Sta=94.7,116.8
XS Rating Curve= 0 ,0
Exp/Cntr(USF)=0,0
Exp/Cntr=0.3,0.1

Type RM Length L Ch R = 1 ,18893   ,469.4,480.2,493.2
XS GIS Cut Line= 3
2208015.34453998395799.958880655 2208320.2987944395945.590096034
2208388.75791274396015.293925617
#Sta/Elev= 30
       0 2355.85    18.7  2351.2    49.7 2338.18    61.5  2335.3    82.5 2333.48
   103.5 2334.04   118.5  2333.5   133.9 2334.72   147.2 2334.96   151.6    2334
   157.5 2331.36   166.5 2329.49   169.5 2329.01   190.5 2329.51     207 2333.17
   218.1 2331.87   238.5  2332.8     272 2332.15   280.5 2331.24   299.9 2332.65
   313.5 2330.44   320.1 2331.54   328.9 2335.32   354.2  2333.8   360.6 2335.69
     372 2342.59     380  2346.4   410.3  2353.7   425.2 2359.11   435.6 2361.41
#Mann= 3 ,-1,0
       0      .1       0   166.5    .045       0   190.5      .1       0
#XS Ineff= 2 , 0
          141.97 2339.85  331.55         2338.19
Permanent Ineff=
       F       F
Bank Sta=166.5,190.5
XS Rating Curve= 0 ,0
Exp/Cntr(USF)=0,0
Exp/Cntr=0.3,0.1

Type RM Length L Ch R = 1 ,18413   ,333.8,334.2,336.2
XS GIS Cut Line= 3
2207777.86350903395993.4314433942207889.58191936396134.549435385
 2207991.0104761396358.721245578
#Sta/Elev= 30
       0 2345.35    25.2 2330.32    32.8 2327.91      47 2326.12    55.6 2325.95
    81.1 2328.94     117 2328.84   175.2 2330.55     190 2329.04   200.4 2326.97
   217.2 2327.72   239.9 2327.56   256.5 2324.57   262.5 2322.75   268.6 2322.41
   274.6 2323.23   286.7  2326.2   295.8  2326.5   305.8 2325.96   314.6 2324.46
   323.4  2324.9     332 2322.91   341.5  2322.5   356.2 2323.04   359.3  2324.1
   365.3 2328.53   380.4 2342.51     398 2349.52   407.6 2352.61     426 2357.12
#Mann= 3 ,-1,0
       0      .1       0     332    .045       0   356.2      .1       0
#XS Ineff= 2 , 0
          293.24 2331.57
Permanent Ineff=
       F       F
Bank Sta=332,356.2
XS Rating Curve= 0 ,0
Exp/Cntr(USF)=0,0
Exp/Cntr=0.3,0.1

Type RM Length L Ch R = 1 ,18079   ,332.9,308.4,284.8
XS GIS Cut Line= 3
2207537.84257069396196.5857054132207613.90825773396303.077667276
2207671.99478239396480.103266218
#Sta/Elev= 30
       0 2333.89     5.6 2332.77    20.4 2330.87    42.2 2327.34      48 2325.94
    59.1 2322.51      68 2320.56    73.8 2319.76    93.9  2318.9     104 2320.23
   116.8 2323.02   133.1 2323.61   141.5 2323.14   153.3 2321.61   162.5 2319.31
   172.4 2318.16   183.6  2317.8   210.4 2318.04   217.3 2319.06   234.1 2319.26
   238.9 2320.71   246.7 2322.38     251 2324.17   259.4 2328.72   268.5  2334.9
   280.4 2343.93   284.6 2345.96   288.8 2346.93   301.5 2347.69   317.2 2347.48
#Mann= 3 ,-1,0
       0      .1       0   172.4    .045       0   210.4      .1       0
Bank Sta=172.4,210.4
XS Rating Curve= 0 ,0
Exp/Cntr(USF)=0,0
Exp/Cntr=0.3,0.1

Type RM Length L Ch R = 1 ,17770   ,243.5,231.3,217.3
XS GIS Cut Line= 2
2207338.68877188396499.4654411022207606.99319527396599.042340506
#Sta/Elev= 30
       0 2359.71     4.9  2353.9    11.8 2346.59    21.2 2335.89    22.9 2333.79
    27.2 2327.65    30.5  2323.8    39.4 2314.61      40 2314.07   41.11 2313.68
    42.9 2312.92    44.3 2312.65    74.1 2312.75    82.7 2313.19    86.9 2313.71
    95.5 2316.52    99.7 2317.42     104 2317.72   111.4  2317.8     121 2317.49
   138.1 2318.78   150.9 2318.55   159.4 2317.84   163.7 2317.91   180.8 2320.33
     185 2320.55   196.4 2320.36   226.5 2320.79   261.8 2323.27   286.2 2325.87
#Mann= 3 ,-1,0
       0      .1       0   41.11    .045       0    86.9      .1       0
#XS Ineff= 2 , 0
                          107.83         2320.26
Permanent Ineff=
       F       F
Bank Sta=41.11,86.9
XS Rating Curve= 0 ,0
Exp/Cntr(USF)=0,0
Exp/Cntr=0.3,0.1

Type RM Length L Ch R = 1 ,17539   ,153.7,153.6,154.3
XS GIS Cut Line= 2
2207299.96442211396759.4717895472207590.39704537396730.428527221
#Sta/Elev= 30
       0 2367.94     8.3 2361.87    28.4  2344.4    38.8 2333.29    44.4 2327.71
    48.5 2323.99    52.5 2320.79    60.5 2315.37      732309.172    76.6 2308.25
    80.6  2307.9    96.7 2307.87   112.8 2307.32   124.8 2308.86   132.9 2309.66
   136.9 2310.61   148.9 2312.63   152.1 2312.82   162.9 2312.39   173.1 2312.38
   181.1 2313.06   185.1  2313.1   189.1 2312.34   201.2 2312.55   213.3 2313.48
   225.3 2316.72   229.3 2317.05   253.5 2316.42   273.6 2317.22   291.9 2318.75
#Mann= 3 ,-1,0
       0      .1       0      73    .045       0   124.8      .1       0
#XS Ineff= 2 , 0
                          153.46         2316.89
Permanent Ineff=
       F       F
Bank Sta=73,124.8
XS Rating Curve= 0 ,0
Exp/Cntr(USF)=0,0
Exp/Cntr=0.3,0.1

Type RM Length L Ch R = 1 ,17386   ,220,225.5,225.9
XS GIS Cut Line= 2
 2207284.7512847396915.752201113 2207602.8441578396882.559901311
#Sta/Elev= 30
       0 2333.17    27.6    2323    31.6 2321.73    39.6 2319.82    47.7 2318.22
    87.9 2314.01    91.9 2311.93    95.9 2307.54     100 2306.07     104 2305.21
   108.7    2305   140.2 2306.03   152.2 2306.47   164.3 2306.35   180.4 2307.51
   184.4 2307.24   192.5 2307.41   196.5 2307.59   204.5 2308.81   208.5 2308.85
   216.6 2307.63   228.7 2308.99   248.8 2307.91   260.8 2308.87   264.9 2309.71
   272.9 2312.14   278.6 2313.21     293  2314.5   300.4 2314.67   319.8 2316.43
#Mann= 3 ,-1,0
       0      .1       0     100    .045       0   140.2      .1       0
#XS Ineff= 2 , 0
                          200.73          2314.6
Permanent Ineff=
       F       F
Bank Sta=100,140.2
XS Rating Curve= 0 ,0
Exp/Cntr(USF)=0,0
Exp/Cntr=0.3,0.1

Type RM Length L Ch R = 1 ,17160   ,206.3,233.8,252.6
XS GIS Cut Line= 5
2207222.51572257396973.838725765 2207351.1358843397084.479725104
2207403.09406487397109.4867534312207566.34024542397118.251649031
2207608.60961809397159.827731719
#Sta/Elev= 30
       0 2328.52    29.1 2315.29    43.3 2310.92    54.6 2309.08     100 2306.38
   160.5 2310.14     171 2309.49   188.6 2305.04   194.9  2304.2   201.9 2304.28
   215.9 2306.56   224.9 2306.62   231.9 2306.02   244.4 2302.65   252.4 2301.65
   268.5 2302.62 275.0222302.109   292.7 2300.78   304.5 2300.96 307.6262301.688
   315.5 2303.87   320.5 2304.39   336.6 2302.92   340.6 2303.82   348.6 2307.58
   356.6  2313.6   372.6 2328.73   399.8 2350.36   411.1 2356.94   450.1  2376.5
#Mann= 3 ,-1,0
       0      .1       0 275.022    .045       0 307.626      .1       0
#XS Ineff= 2 , 0
          221.13 2313.07
Permanent Ineff=
       F       F
Bank Sta=275.022,307.626
XS Rating Curve= 0 ,0
Exp/Cntr(USF)=0,0
Exp/Cntr=0.3,0.1

Type RM Length L Ch R = 1 ,16926   ,237.1,256.8,268.8
XS GIS Cut Line= 2
2207189.32342277397018.0951255012207359.43395925397345.869086041
#Sta/Elev= 30
       0 2317.88      17 2310.79      40  2305.8    62.1 2303.99    81.5 2303.36
    89.1 2303.38   111.6 2305.81   129.7 2305.28   138.7 2303.38   147.7 2298.98
   152.2 2297.45   162.5 2295.54   165.7 2295.39   174.7 2296.76   179.4 2298.28
   192.8 2298.63   205.9 2297.49   215.3 2297.32   224.3  2298.6   242.3 2299.34
   255.8 2298.71   272.42296.085   287.4 2295.23   304.1 2296.29     310 2298.22
   318.9 2302.28     328 2307.59   341.5 2318.38   360.4 2336.15   369.3 2343.47
#Mann= 3 ,-1,0
       0      .1       0   272.4    .045       0   304.1      .1       0
#XS Ineff= 2 , 0
          177.57 2305.69
Permanent Ineff=
       F       F
Bank Sta=272.4,304.1
XS Rating Curve= 0 ,0
Exp/Cntr(USF)=0,0
Exp/Cntr=0.3,0.1

Type RM Length L Ch R = 1 ,16669   ,279.6,278.4,273.5
XS GIS Cut Line= 2
2207149.21606051397047.1383878272207064.85229852397354.167160991
#Sta/Elev= 30
       0 2311.68    18.7 2307.03    43.6 2302.63    60.2  2300.4    68.5 2298.71
    76.8 2298.11    89.2 2297.98    97.5 2298.33   103.4 2297.93   118.3 2295.65
   130.7  2292.2   134.9 2291.74   143.2 2292.05   151.5 2293.75   159.7 2293.56
   176.3 2294.35   180.5  2294.2   192.9 2290.78   197.1 2290.11   213.7 2288.53
   226.1 2289.27   238.6 2288.81   245.5 2289.93   246.9 2290.33     251 2293.17
   259.6 2299.54   271.8 2309.26   285.6  2319.2   300.8 2328.51   318.4 2338.12
#Mann= 3 ,-1,0
       0      .1       0   197.1    .045       0   245.5      .1       0
Bank Sta=197.1,245.5
XS Rating Curve= 0 ,0
Exp/Cntr(USF)=0,0
Exp/Cntr=0.3,0.1

Type RM Length L Ch R = 1 ,16391   ,324.4,327.7,336.7
XS GIS Cut Line= 2
2206863.01987799 396990.110973362206804.93335334 397309.58685895
#Sta/Elev= 30
       0 2331.65    15.3 2321.25    39.7 2299.12    51.9 2290.17      56  2288.1
      60 2287.53    80.4 2287.92   104.8 2287.06   118.6 2287.83   133.2  2287.2
   141.3 2288.08   149.5 2288.13   157.6 2287.57   161.7 2288.12   166.8 2288.19
   186.1 2286.81   204.6 2283.24   226.7 2282.17   230.8  2282.3   235.6  2283.2
   238.9 2284.48   242.5 2286.72   249.3 2291.94   255.2 2295.51   263.3 2301.11
   275.5 2306.55   287.7 2313.36   295.8 2317.22     308 2323.79   324.7 2331.87
#Mann= 3 ,-1,0
       0      .1       0   204.6    .045       0   235.6      .1       0
#XS Ineff= 2 , 0
          167.61 2299.59
Permanent Ineff=
       F       F
Bank Sta=204.6,235.6
XS Rating Curve= 0 ,0
Exp/Cntr(USF)=0,0
Exp/Cntr=0.3,0.1

Type RM Length L Ch R = 1 ,16063   ,216.2,201.6,185.3
XS GIS Cut Line= 3
2206608.45817624396914.3691886212206503.34922687397110.756962447
2206506.11525186397243.526161653
#Sta/Elev= 30
       0 2323.63     7.7 2318.97    21.3 2312.33    25.9 2310.78    30.4 2308.01
    46.6 2294.71    58.4 2287.75    71.2 2283.65    84.9 2281.23    96.9 2280.33
   107.5  2281.3   129.4  2281.2   139.3 2278.72   157.4 2277.05   175.6 2277.41
   190.12278.896   197.3  2280.9   202.8 2281.35   249.2 2280.13   265.2 2281.74
   273.2 2284.65   289.2 2293.02   293.2 2296.57   301.2 2306.68   309.2 2318.21
   313.2  2322.6   325.2 2332.11   337.2 2339.25   349.2 2350.74   355.5 2354.58
#Mann= 3 ,-1,0
       0      .1       0   139.3    .045       0   190.1      .1       0
#XS Ineff= 2 , 0
                          235.94         2289.47
Permanent Ineff=
       F       F
Bank Sta=139.3,190.1
XS Rating Curve= 0 ,0
Exp/Cntr(USF)=0,0
Exp/Cntr=0.3,0.1

Type RM Length L Ch R = 1 ,15862   ,195.8,196.2,192.8
XS GIS Cut Line= 2
2206330.47266541396936.4973884892206369.19701517 397225.54699926
#Sta/Elev= 30
       0 2307.32    20.9 2298.04    28.9 2292.94      41 2283.06    45.1 2280.52
    53.2 2278.35    61.2 2273.71    65.3 2272.15    69.3 2271.58    85.4 2272.67
    93.5 2273.92   101.6 2277.91   105.3 2278.17   109.7 2277.92   125.8  2275.6
   137.4 2275.87     146 2276.74   158.7  2276.1   170.2 2276.04   178.3 2275.04
   186.3 2274.79   190.4 2275.05   194.3  2276.1   198.4 2277.35   202.5 2279.39
   222.8 2295.86   233.5 2300.73   247.7 2309.06   278.4 2325.18   291.6 2333.23
#Mann= 3 ,-1,0
       0      .1       0    61.2    .045       0    93.5      .1       0
#XS Ineff= 2 , 0
                          106.48         2281.16
Permanent Ineff=
       F       F
Bank Sta=61.2,93.5
XS Rating Curve= 0 ,0
Exp/Cntr(USF)=0,0
Exp/Cntr=0.3,0.1

Type RM Length L Ch R = 1 ,15665   ,203.8,203.6,204
XS GIS Cut Line= 2
2206146.53200401396975.2217382572206193.55442873397224.163986769
#Sta/Elev= 30
       0 2294.26    22.3 2284.95    38.6 2279.46    42.7 2278.34    46.8 2277.37
      59 2275.43    67.1 2274.88    75.3 2275.15    79.3 2274.61   105.8 2268.73
   111.9 2267.79   115.8 2267.75     120 2267.84   129.8 2268.95   144.5 2270.09
   148.5  2270.2   156.7 2269.61   160.8 2270.76   164.8 2273.16   168.9 2276.01
     173 2278.19   181.3 2280.26   185.2 2281.44   193.3 2285.27   201.5 2288.75
   213.7 2294.86   221.8 2298.68   231.3 2302.52   246.2 2309.24   253.3 2312.83
#Mann= 3 ,-1,0
       0      .1       0   105.8    .045       0   129.8      .1       0
Bank Sta=105.8,129.8
XS Rating Curve= 0 ,0
Exp/Cntr(USF)=0,0
Exp/Cntr=0.3,0.1

Type RM Length L Ch R = 1 ,15462   ,205,201.5,197.3
XS GIS Cut Line= 2
2205950.14423018397009.7970505512205995.78364241397262.888336537
#Sta/Elev= 30
       0 2300.55    11.4 2292.42    27.8 2282.16    31.9 2279.99    44.1 2271.52
    48.1 2269.12    52.2 2267.36    56.3 2266.09    60.3 2265.53    64.4  2265.9
    72.5 2267.95    83.9 2268.76    92.9 2270.34     101 2269.37   109.1 2266.12
   113.2 2264.91   117.2 2264.19   129.4 2263.32   149.8  2263.8   158.72264.773
     162 2265.53     166 2267.59   174.1 2273.09   178.2 2275.03   182.3 2275.78
   198.5 2277.23   206.7  2279.1   214.8  2281.8   235.1 2291.43   257.2 2304.05
#Mann= 3 ,-1,0
       0      .1       0   113.2    .045       0   158.7      .1       0
#XS Ineff= 2 , 0
           94.99 2272.99
Permanent Ineff=
       F       F
Bank Sta=113.2,158.7
XS Rating Curve= 0 ,0
Exp/Cntr(USF)=0,0
Exp/Cntr=0.3,0.1

Type RM Length L Ch R = 1 ,15260   ,194.2,199.2,205.3
XS GIS Cut Line= 2
 2205746.8413939 397096.926837532205824.29009343397300.229673814
#Sta/Elev= 30
       0  2279.3     4.6 2275.64      15 2266.25    17.4 2264.53    21.7 2262.39
      26 2261.94    34.5 2263.66    38.8 2263.72    47.4 2263.07    51.6 2262.52
    55.9 2261.62    60.2 2260.15    63.2 2259.59      73 2259.23    90.2 2259.32
    97.3 2259.61     103 2260.45   115.8  2263.9   128.7 2263.87   137.2 2263.24
   141.5 2263.47   145.8 2264.25   149.8 2265.43   154.4 2267.28   158.6 2267.84
   171.5 2268.68   175.8 2270.07   194.8 2277.65   205.6 2282.83   217.6 2289.19
#Mann= 3 ,-1,0
       0      .1       0    63.2    .045       0    97.3      .1       0
#XS Ineff= 2 , 0
           37.46 2266.81
Permanent Ineff=
       F       F
Bank Sta=63.2,97.3
XS Rating Curve= 0 ,0
Exp/Cntr(USF)=0,0
Exp/Cntr=0.3,0.1

Type RM Length L Ch R = 1 ,15061   ,211.1,208.9,205.5
XS GIS Cut Line= 4
2205565.66675748397094.1608125462205583.64591987397254.590261587
2205593.32700731397344.486073549 2205612.6891822397379.061385843
#Sta/Elev= 30
       0 2294.01    11.1 2290.78    23.2 2286.25    35.2 2282.92    39.3 2281.22
    47.3 2276.22    59.3 2264.77    63.4 2262.06    75.5 2259.36    84.6 2255.75
    99.6 2254.76   111.7 2255.06   115.7 2255.79   123.8 2258.71   127.8  2259.4
   135.9 2259.32   143.9 2260.72     152 2261.38   168.1 2261.31   192.2 2258.65
   200.6 2259.33   212.3 2262.46   216.3 2263.05   224.4 2263.52   232.4 2263.28
   240.5 2264.18   248.5 2265.91   261.8 2270.57   275.6 2277.19   291.5 2286.89
#Mann= 3 ,-1,0
       0      .1       0    84.6    .045       0   115.7      .1       0
#XS Ineff= 2 , 0
                           158.2         2274.84
Permanent Ineff=
       F       F
Bank Sta=84.6,115.7
XS Rating Curve= 0 ,0
Exp/Cntr(USF)=0,0
Exp/Cntr=0.3,0.1

Type RM Length L Ch R = 1 ,14852   ,308.9,318.9,328.6
XS GIS Cut Line= 3
2205347.15078379397128.7361248392205403.85429595  397352.7841485
2205381.72609608397446.828997937
#Sta/Elev= 30
       0 2282.91    27.5 2275.05    37.6  2272.7    41.7  2271.3    47.3 2268.01
    54.1 2263.04    62.3 2257.78    78.9 2251.49    86.8 2250.84   103.6 2251.04
   109.9 2251.59     116    2253   120.1 2254.42   132.9  2255.6   144.9    2256
   153.1 2255.79   157.2 2255.18   161.4 2253.96   165.5 2253.68   173.8 2254.61
   194.4 2255.66   239.7  2259.5   264.4 2260.14   276.7 2264.46   284.4 2267.71
   291.1 2271.08   301.4 2276.98   313.7 2284.99     321 2288.91   327.7  2293.4
#Mann= 3 ,-1,0
       0      .1       0    78.9    .045       0   109.9      .1       0
Bank Sta=78.9,109.9
XS Rating Curve= 0 ,0
Exp/Cntr(USF)=0,0
Exp/Cntr=0.3,0.1

Type RM Length L Ch R = 1 ,14533   ,252.8,267.1,284.8
XS GIS Cut Line= 4
2205212.49521068397112.0319945052205068.34499948397288.071501276
2205060.67571583397316.5574119762205003.91282606397371.104701651
#Sta/Elev= 30
       0 2271.82    13.1 2264.65    27.3 2257.45    32.5 2255.33    37.7 2253.94
    42.8 2253.12    60.7 2252.98    69.3 2252.22    82.6 2252.71    97.7 2254.14
   110.1 2253.57   120.4 2254.47   141.1 2251.52   168.7 2251.52   180.1 2250.93
   194.3 2248.96   213.5 2247.48   222.8 2245.49229.51192245.038   249.4 2244.11
 254.146 2245.03   263.7 2250.25   269.5 2254.14     281  2267.3   288.9 2274.91
   300.3 2284.94   308.7 2292.85   317.2 2299.72   325.7 2307.83   335.8 2316.25
#Mann= 3 ,-1,0
       0      .1       0229.5119    .045       0 254.146      .1       0
Bank Sta=229.5119,254.146
XS Rating Curve= 0 ,0
Exp/Cntr(USF)=0,0
Exp/Cntr=0.3,0.1

Type RM Length L Ch R = 1 ,14266   ,232.9,230.9,221.1
XS GIS Cut Line= 3
2205106.50661023397005.6480130752204850.64929925397116.289012414
2204811.92494949397167.460474608
#Sta/Elev= 30
       0 2281.99    28.7 2267.33    46.1 2259.26    56.2 2255.56    76.6 2249.24
    80.5 2248.48    92.7 2246.87    98.8 2246.39   107.9 2246.22   115.8 2244.97
   123.1 2244.67   133.3 2244.93   147.5 2244.62   155.1 2243.09   168.7 2240.85
   174.8  2239.9   181.2 2239.41   194.3 2239.31   214.4 2239.66   220.4  2240.3
  222.68 2240.88   224.8 2241.58   229.2 2243.86   233.5 2246.62   246.6 2254.23
   259.7 2262.79   277.1 2275.16   315.4 2303.51   329.3 2312.29   342.9 2321.33
#Mann= 3 ,-1,0
       0      .1       0   168.7    .045       0  222.68      .1       0
Bank Sta=168.7,222.68
XS Rating Curve= 0 ,0
Exp/Cntr(USF)=0,0
Exp/Cntr=0.3,0.1

Type RM Length L Ch R = 1 ,14035   ,278.2,269.3,259.2
XS GIS Cut Line= 2
2204946.07716118396805.1112017742204687.45382523 396969.68968829
#Sta/Elev= 30
       0 2275.41    35.4 2259.24    44.9 2256.36    59.1 2250.78    73.4 2244.59
    82.9 2241.12    92.3  2239.5   108.6 2239.34   130.3 2240.42     135 2240.17
   144.5 2234.89     154 2234.03   169.5 2234.13  179.61 2234.89   187.2 2237.99
   191.9 2238.89   195.6 2239.08   220.4 2235.34   223.6 2235.56   240.7 2241.76
   248.8 2246.32   259.3 2258.39     263 2262.12   272.5 2268.05   282.5 2272.66
   285.4 2274.72   288.3 2277.92   291.5 2282.12   298.1 2289.36   306.5 2294.15
#Mann= 3 ,-1,0
       0      .1       0   144.5    .045       0  179.61      .1       0
#XS Ineff= 2 , 0
          130.93 2243.91  193.24         2243.83
Permanent Ineff=
       F       F
Bank Sta=144.5,179.61
XS Rating Curve= 0 ,0
Exp/Cntr(USF)=0,0
Exp/Cntr=0.3,0.1

Type RM Length L Ch R = 1 ,13766   ,220.2,212,194
XS GIS Cut Line= 3
2204697.13491267396554.7859407712204607.23910071396780.216976923
2204583.72788835 396921.28425108
#Sta/Elev= 30
       0 2281.66    24.1 2267.71    48.8  2256.6    54.3 2253.66    64.2 2247.27
    75.8 2237.52    80.1 2234.68    88.7 2232.32   107.3 2233.97   118.8 2232.93
     135 2230.48   144.7 2229.78   153.8 2230.54   170.5  2231.1   187.3 2232.94
   207.8 2233.18   218.1 2235.73   229.4    2235   235.1 2235.84   247.7 2235.27
   263.9 2235.73     268 2235.39   276.1 2232.11   280.2 2231.39   312.6 2234.32
   316.7  2235.6   320.7  2238.3   328.8 2246.21   332.9 2248.85   385.7 2279.55
#Mann= 3 ,-1,0
       0      .1       0     135    .045       0   153.8      .1       0
Bank Sta=135,153.8
XS Rating Curve= 0 ,0
Exp/Cntr(USF)=0,0
Exp/Cntr=0.3,0.1

Type RM Length L Ch R = 1 ,13554   ,217.2,212.7,209.3
XS GIS Cut Line= 3
2204419.14940184396556.1689532632204456.49073911396717.981414795
2204477.23592649396910.220151146
#Sta/Elev= 30
       0 2270.48    54.4 2228.87    58.5 2227.52    62.6  2226.9    83.1 2227.41
     116 2226.61   124.2 2227.52   128.3 2230.07   132.4 2231.43   136.5 2231.68
   148.8 2230.94   169.3 2232.76   201.5 2229.69   213.5 2230.79   225.6 2229.64
   233.7 2230.72   241.7 2228.83   245.7 2228.42   249.7 2228.44   257.8 2229.49
   277.9 2230.14     286 2231.58     294 2232.33   300.8 2234.35   310.1 2239.26
   318.1 2244.57   326.2 2249.25   350.4 2265.63   354.3 2268.43   359.4 2272.83
#Mann= 3 ,-1,0
       0      .1       0    83.1    .045       0   124.2      .1       0
#XS Ineff= 1 ,-1
  167.89  214.76 2235.83
Permanent Ineff=
       F
Bank Sta=83.1,124.2
XS Rating Curve= 0 ,0
Exp/Cntr(USF)=0,0
Exp/Cntr=0.3,0.1

Type RM Length L Ch R = 1 ,13341   ,155.9,155.5,156.5
XS GIS Cut Line= 3
2204189.56932821396615.6384904072204282.23116515396784.366014398
2204326.48756489396936.497388489
#Sta/Elev= 30
       0 2279.33    20.7 2268.42    30.3  2261.6    38.3 2257.59    47.4 2250.25
      52 2247.14    61.1 2239.76    70.2  2231.6    74.8 2228.38    96.8 2221.23
   106.7 2220.76   115.8  2221.1   129.7 2223.42   152.4 2223.02     166 2223.87
     171 2224.43   179.7 2227.12   193.3 2228.85     210 2227.69   222.5 2225.45
   230.8 2224.84   247.5  2224.7     260 2226.83   264.2 2226.56   272.5 2224.66
   276.7 2224.41   281.9 2225.09   289.2 2227.56   317.3 2247.91   350.9 2268.18
#Mann= 3 ,-1,0
       0      .1       0    96.8    .045       0   115.8      .1       0
Bank Sta=96.8,115.8
XS Rating Curve= 0 ,0
Exp/Cntr(USF)=0,0
Exp/Cntr=0.3,0.1

Type RM Length L Ch R = 1 ,13186   ,170.4,170.1,170.3
XS GIS Cut Line= 3
2204051.26807904396686.1721274862204152.22799093396861.814713935
2204175.73920329396972.455713274
#Sta/Elev= 30
       0 2276.27    43.9 2251.96      50 2249.39    72.7 2231.65      79 2226.32
    81.9 2224.15    86.5 2221.82    91.1 2220.75   109.6  2218.3     1302217.724
   137.6 2216.78   143.5 2216.62   151.1 2216.95   154.3 2218.01   160.3 2220.67
   162.4 2221.07   164.9 2221.16   178.8 2218.94   181.6 2219.32     188  2221.8
   192.6 2222.56   214.2 2222.14     251 2219.39   260.1 2219.64   263.3 2220.29
   279.6 2227.09   287.8 2231.05   300.1 2238.17   308.3 2244.32   315.7 2249.08
#Mann= 3 ,-1,0
       0      .1       0     130    .045       0   154.3      .1       0
Bank Sta=130,154.3
XS Rating Curve= 0 ,0
Exp/Cntr(USF)=0,0
Exp/Cntr=0.3,0.1

Type RM Length L Ch R = 1 ,13016   ,143.6,146,146.7
XS GIS Cut Line= 2
2203919.88189232396799.5791518072204062.33217897397045.755375336
#Sta/Elev= 30
       0 2255.25     7.2 2251.99    15.7 2248.69      25 2245.77    51.2 2235.31
    62.9 2229.78    77.5 2221.57    88.4 2214.83    92.1 2213.38    94.3 2213.04
   112.4 2214.12   135.9 2214.09   141.9 2214.77   152.3 2215.89   160.3 2217.44
   168.2 2217.62   177.5 2216.27   188.7 2218.17   194.6 2218.87     201 2219.11
     212 2218.52   223.7 2218.55   228.3    2219   232.7 2219.93   237.5 2221.44
   242.2 2223.34   251.4 2227.74   260.6 2232.97   269.9 2237.84   284.4 2247.19
#Mann= 3 ,-1,0
       0      .1       0    88.4    .045       0   141.9      .1       0
Bank Sta=88.4,141.9
XS Rating Curve= 0 ,0
Exp/Cntr(USF)=0,0
Exp/Cntr=0.3,0.1

Type RM Length L Ch R = 1 ,12870   ,188.8,191.8,195
XS GIS Cut Line= 2
2203791.95707777396845.4442734882203928.90857151 397141.25949998
#Sta/Elev= 30
       0 2258.07    12.9 2252.41    26.2 2247.68      35 2245.33    48.2 2240.34
    57.6 2236.26    72.3  2231.6    83.5 2226.01    99.4 2216.01   105.5 2212.77
   109.9 2211.64   117.5    2211   140.8 2210.31   150.6 2210.43   158.4 2211.13
     176 2215.92   177.7 2216.06   189.8 2215.98   202.5 2214.78   211.3 2214.96
   228.8 2213.97     235 2214.29   246.5 2213.58     251 2214.42   259.1 2217.54
   276.6 2226.26   286.2 2230.56   308.3 2243.02   317.1  2248.4     326 2254.44
#Mann= 3 ,-1,0
       0      .1       0   117.5    .045       0   158.4      .1       0
Bank Sta=117.5,158.4
XS Rating Curve= 0 ,0
Exp/Cntr(USF)=0,0
Exp/Cntr=0.3,0.1

Type RM Length L Ch R = 1 ,12678   ,252.2,254.7,261.6
XS GIS Cut Line= 2
2203629.44926906396900.539063704 2203723.4941185397240.760136669
#Sta/Elev= 30
       0  2254.6    12.5 2246.61    21.4 2241.42    42.2 2231.14    50.5 2227.45
    54.6  2224.8    62.9 2220.56    75.4 2213.01    79.5 2211.57    87.3 2209.84
      92 2209.61     106 2207.07   112.7 2206.63     136 2207.12   162.5 2207.57
   166.7 2208.53   170.8 2210.52   179.1 2212.46   183.3 2212.27   191.3 2212.66
   195.7 2212.26   204.3 2212.96   232.2 2210.62   237.2 2209.85   241.4 2210.15
   282.9 2216.01   295.3 2218.95   307.8 2223.13   329.7  2232.8     353 2245.02
#Mann= 3 ,-1,0
       0      .1       0     106    .045       0     136      .1       0
Bank Sta=106,136
XS Rating Curve= 0 ,0
Exp/Cntr(USF)=0,0
Exp/Cntr=0.3,0.1

Type RM Length L Ch R = 1 ,12423   ,174.6,181.6,189.4
XS GIS Cut Line= 3
2203402.63522041396928.1993135382203410.93329536397164.694449624
2203383.27304553397283.633523913
#Sta/Elev= 30
       0  2248.4      13 2241.64      33 2232.35      57 2219.76      73 2207.37
      81 2202.92    84.52201.429      89 2200.87      97 2200.67     109 2201.08
   133.1 2203.59   149.1 2204.47     161 2204.06   173.1 2204.53   189.1 2202.13
   207.4 2201.61   213.1 2202.55   217.1 2204.62   221.1 2205.48   229.1  2205.7
   245.4 2205.67   253.6 2203.59     270 2203.11   278.2 2202.08   290.5 2202.74
   294.6 2203.95   303.2  2208.5   322.6 2219.79     336 2225.53   358.8 2237.94
#Mann= 3 ,-1,0
       0      .1       0    84.5    .045       0     109      .1       0
Bank Sta=84.5,109
XS Rating Curve= 0 ,0
Exp/Cntr(USF)=0,0
Exp/Cntr=0.3,0.1
